--- GEORGESCK.prj (project) ---

Proj Title=GEORGESCK
Current Plan=p01
Default Exp/Contr=0,0
English Units
Geom File=g01
Flow File=f01
Plan File=p01
BEGIN DESCRIPTION:
END DESCRIPTION:
DSS Export Rating Curves= 0
DSS Export Rating Curve Sorted= 0
DSS Export Volume Flow Curves= 0
DXF OffsetX= 0
DXF OffsetY= 0
DXF ScaleX= 0
DXF ScaleY= 0

--- GEORGESCK.p01 (plan) ---

Plan Title=Floodplain
Program Version=4.00
Geom File=g01
Flow File=f01
K Sum by GR=0
Std Step Tol=0.01
Critical Tol=0.01
Num of Std Step Trials=20
Max Error Tol=0.3
Flow Tol Ratio=0.001
Split Flow NTrial=30
Split Flow Tol=0.02
Split Flow Ratio=0.02
Log Output Level=0
Friction Slope Method=1
Unsteady Friction Slope Method=2
Unsteady Bridges Friction Slope Method=1
Global Log Level=0
CheckData=False
Run HTab=0
Run UNet=0
Run PostProcess=0
UNET Theta=0
UNET Theta Warmup=0
UNET ZTol=0
UNET ZSATol=0
UNET MxIter=0
UNET MaxInSteps=0
UNET DtIC=0
UNET DtMin=0
UNET MaxCRTS=0
UNET WFStab=0
UNET SFStab=0
UNET WFX=0
UNET SFX=0
UNET DSS MLevel=0
UNET DZMax Abort=0
UNET Convert EG Bridges=0
UNET Use Existing IB Tables=0
UNET Froude Limit=0
UNET Froude Power=0
Write IC File=0
Echo Input=False
Echo Output=False
Write Detailed=0

--- GEORGESCK.f01 (steady flow) ---

Flow Title=NFF Regression Equation
Program Version=4.10
Number of Profiles= 1
Profile Names=P100yr
River Rch & RM=GEORGESCK,Main            ,9388.3
      59
River Rch & RM=GEORGESCK,Main            ,8260.4
     190
River Rch & RM=GEORGESCK,Main            ,7649.4
     227
River Rch & RM=GEORGESCK,Main            ,6286.7
     292
River Rch & RM=GEORGESCK,Main            ,5790.3
     342
River Rch & RM=GEORGESCK,Main            ,4649.8
     496
River Rch & RM=GEORGESCK,Main            ,2852.1
     547
River Rch & RM=GEORGESCK,Main            ,775.7
     585
Boundary for River Rch & Prof#=GEORGESCK,Main            , 1
Up Type= 0
Dn Type= 1
Dn Known WS=721.2
DSS Import GetInterval= 0
DSS Import GetPeak= 0
DSS Import FillOption= 0

--- GEORGESCK.g01 (geometry) ---

Geom Title=USGS 10m DEM
Program Version=4.10

River Reach=GEORGESCK       ,Main
Reach XY= 30
     1814231.611      461939.805     1814420.586       462274.05
     1814793.071      462652.387     1814826.836      462921.967
     1814719.865      463367.346     1814751.142      463479.606
     1814629.587      463600.419     1814613.224      463852.537
     1814509.475      463968.495      1814340.09      464747.989
     1814168.633      464983.825     1814038.543      465295.079
     1814021.189      465413.368     1813683.781      465951.134
     1812974.552      466449.117      1812656.09      466791.368
     1812408.694      466899.441     1812286.298      467116.889
     1812106.323      467315.263     1811864.423       467674.18
     1811798.017      467714.545     1811781.805      467840.698
     1811575.073      468234.013     1811343.817      468504.891
     1811195.152      468515.326     1811028.111      468821.007
     1811048.243      468967.296     1810902.184      469077.826
     1810849.314      469182.682     1810641.414      469401.866

Type RM Length L Ch R = 1 ,9388.3  ,337.8,339,340.2
XS GIS Cut Line= 2
     1814141.848      462024.479     1814393.584      461907.291
#Sta/Elev= 25
       0 1145.29    19.2 1141.08    28.7 1139.14    47.9 1135.63    57.4 1133.82
      67 1131.86    76.6  1129.6    86.2 1126.59    95.8  1121.5   105.3 1115.39
   114.9 1111.44   124.5 1111.99     134 1116.02   143.6 1121.16   153.2 1125.56
   162.8 1129.07   172.4 1132.27   181.9 1135.29   201.1 1141.17   210.6 1144.18
   220.2 1147.28   229.8  1150.5   239.4 1153.89     249 1157.42   277.7 1168.28
#Mann= 3 , 0 , 0
       0      .1       0   114.9    .045       0   124.5      .1       0
Bank Sta=114.9,124.5
XS Rating Curve= 0 ,0
Exp/Cntr=0.3,0.1

Type RM Length L Ch R = 1 ,9049.3  ,304,298.5,293
XS GIS Cut Line= 3
     1814302.439      462315.277     1814516.833      462227.478
     1814621.709      462152.822
#Sta/Elev= 30
       0 1088.75    38.6 1069.96    48.3 1065.39    57.9 1060.93    67.6 1056.92
    77.2 1054.02    86.9 1052.03   106.2 1048.38   115.6 1047.27   125.5  1047.7
   135.1 1049.81   144.8 1052.56   154.4 1054.94   164.1    1057   173.8 1059.26
   193.1 1064.12   212.4 1069.31   231.7 1074.83   250.1 1082.08   259.3 1085.85
   268.5 1089.41   277.6 1092.49     296  1097.5   305.2 1099.48   314.4 1100.41
   323.6 1100.61   332.8 1100.22     342 1099.42   351.2 1098.16   360.4 1096.57
#Mann= 3 , 0 , 0
       0      .1       0   115.6    .045       0   125.5      .1       0
Bank Sta=115.6,125.5
XS Rating Curve= 0 ,0
Exp/Cntr=0.3,0.1

Type RM Length L Ch R = 1 ,8750.8  ,265.3,268.9,272.2
XS GIS Cut Line= 2
     1814541.154      462536.632     1814753.828      462382.552
#Sta/Elev= 30
       0 1064.22     9.7  1059.4    19.4 1054.89    29.2 1050.41    38.9 1045.79
    48.6 1041.17    58.4 1036.56    68.1 1032.01    77.8 1027.48    87.5 1023.66
    97.3 1021.47      98 1021.43     107 1020.85     113 1021.09   116.7 1021.24
   126.4 1022.18   136.2 1022.98   145.9 1023.58   155.6  1024.1   165.4 1024.57
   175.1 1024.96   184.8 1025.28   194.5 1025.57   204.3 1025.78     214    1026
   223.7 1026.12   233.4 1026.29   243.2 1026.51   252.9 1026.72   262.6 1026.99
#Mann= 3 , 0 , 0
       0      .1       0      98    .045       0     113      .1       0
Bank Sta=98,113
XS Rating Curve= 0 ,0
Exp/Cntr=0.3,0.1

Type RM Length L Ch R = 1 ,8481.9  ,210.1,221.6,232.9
XS GIS Cut Line= 3
     1814723.446      462691.146     1814779.435      462687.239
     1814903.133      462623.437
#Sta/Elev= 23
       0 1028.46     9.4 1024.72    18.7 1020.87    28.1 1016.76    37.4 1012.43
    46.8 1008.27    56.1 1005.37    65.4  1004.3    74.7 1003.74      84 1003.75
    89.7 1004.12    93.2 1004.34   102.5 1005.02   111.8 1005.46   121.1 1005.76
   130.4 1006.02   139.6 1006.24   148.9 1006.47   158.2 1006.72   167.5 1006.92
   176.8 1007.15     186  1007.4   195.3 1007.67
#Mann= 3 , 0 , 0
       0      .1       0    74.7    .045       0    89.7      .1       0
Bank Sta=74.7,89.7
XS Rating Curve= 0 ,0
Exp/Cntr=0.3,0.1

Type RM Length L Ch R = 1 ,8260.4  ,99.7,106.5,110.7
XS GIS Cut Line= 4
     1814744.279      462882.552     1814802.873      462894.271
     1814896.623      462896.875     1815012.508      462831.771
#Sta/Elev= 23
       0 1017.44    17.1 1010.32    34.2 1003.14    42.7  999.48    51.2  995.96
    59.8  992.91    69.1  990.46    78.5  988.86    87.9  988.24    97.3  988.57
     116  989.87   153.5  992.26   172.5  993.78     201  995.75   210.5  996.54
     220  997.85   229.5  999.87     239 1002.35   248.5 1005.22     258 1008.46
   267.5 1012.03     277 1015.74   286.5 1019.71
#Mann= 3 , 0 , 0
       0      .1       0    78.5    .045       0    97.3      .1       0
Bank Sta=78.5,97.3
XS Rating Curve= 0 ,0
Exp/Cntr=0.3,0.1

Type RM Length L Ch R = 1 ,8153.9  ,186.2,189.9,192.9
XS GIS Cut Line= 4
      1814755.13      462973.264     1814806.605      462998.308
     1814846.536      463006.989      1814942.89      463004.385
#Sta/Elev= 24
       0 1003.09     9.5  998.76    19.1  994.48    28.6  990.59    38.2  987.85
    47.7  985.83    57.2  983.85    61.6  983.15    65.4  982.55    73.6     982
    76.6  982.16    81.8  982.43    89.9  983.81    98.1  985.66   107.8  987.81
   117.4  989.59     127  990.79   136.7  990.87   146.3  990.36   155.9  990.66
   165.6   991.9   175.2  993.31   184.9  994.68   194.5  996.22
#Mann= 3 , 0 , 0
       0      .1       0    65.4    .045       0    81.8      .1       0
Bank Sta=65.4,81.8
XS Rating Curve= 0 ,0
Exp/Cntr=0.3,0.1

Type RM Length L Ch R = 1 ,7963.9  ,316.3,314.5,317
XS GIS Cut Line= 3
     1814713.029      463148.177     1814762.508      463179.427
     1814896.623      463227.604
#Sta/Elev= 23
       0  997.73     9.8  993.24    19.5  988.81    29.3  984.56      39  981.31
    48.8  978.67    58.4  976.25      68  974.27    73.4  973.96    77.5  973.73
      87  974.03    96.5  974.43     106     975   115.5  975.68     125  977.15
   134.5  979.68     144  982.83   153.5  986.11     163  989.45   172.5  992.78
     182  996.14   191.5  999.52     201 1002.88
#Mann= 3 , 0 , 0
       0      .1       0      68    .045       0      87      .1       0
Bank Sta=68,87
XS Rating Curve= 0 ,0
Exp/Cntr=0.3,0.1

Type RM Length L Ch R = 1 ,7649.4  ,281.5,272.8,262
XS GIS Cut Line= 4
     1814617.977      463446.354     1814723.446      463469.791
     1814766.414      463488.021     1814843.237      463550.521
#Sta/Elev= 30
       0  997.97     9.8  996.94    19.6  996.14    29.5  995.33    39.3  994.23
    49.1  992.87    58.9  991.51    68.8  990.11    78.6  988.57    88.4   986.3
    98.2  982.56     108   977.1   117.4  970.47   126.7  963.53   129.6  962.83
     136   961.3   144.6  963.33   145.4  963.52   154.7  968.15   163.7  972.52
   172.7  976.45   181.7  980.17   190.7     984   199.7  987.91   208.7  991.83
   217.7   995.8   226.7  999.67   235.8 1003.56   244.8 1007.46   253.8 1011.16
#Mann= 3 , 0 , 0
       0      .1       0   129.6    .045       0   144.6      .1       0
Bank Sta=129.6,144.6
XS Rating Curve= 0 ,0
Exp/Cntr=0.3,0.1

Type RM Length L Ch R = 1 ,7376.5  ,252.6,271.7,290.7
XS GIS Cut Line= 3
     1814541.154       463700.26     1814660.946      463702.864
     1814729.956       463693.75
#Sta/Elev= 24
       0   969.1     9.2  966.97    18.4  964.95    27.6  962.62    36.9  959.65
    46.1  955.86    55.3  950.65    64.5  944.12    73.7  938.79    74.9   938.6
      83   937.3    89.9   939.3    92.2  939.97   101.4  945.43   110.6  950.54
   119.8  954.64   128.5  958.27   137.2  961.76   145.9  965.08   154.6  968.19
   163.3   971.1     172  973.85   180.7  976.55   189.4  979.35
#Mann= 3 , 0 , 0
       0      .1       0    74.9    .045       0    89.9      .1       0
Bank Sta=74.9,89.9
XS Rating Curve= 0 ,0
Exp/Cntr=0.3,0.1

Type RM Length L Ch R = 1 ,7104.8  ,187.4,174.8,161.2
XS GIS Cut Line= 3
     1814489.071      463890.364     1814552.873      463963.281
     1814623.185      463986.718
#Sta/Elev= 21
       0  964.21     9.7  958.73    19.4     951    29.1  942.34    38.8  933.34
    48.4  925.51    56.8  921.72    58.1  921.13    67.8  919.85    71.8  920.43
    77.5  921.25    87.2  923.69    96.9  926.11   106.2  928.75   115.4  931.34
   124.7  934.05     134  936.84   143.2  939.64   152.5  942.48   161.7  945.39
     171  948.34
#Mann= 3 , 0 , 0
       0      .1       0    58.1    .045       0    71.8      .1       0
Bank Sta=58.1,71.8
XS Rating Curve= 0 ,0
Exp/Cntr=0.3,0.1

Type RM Length L Ch R = 1 ,6930    ,223.9,226.9,230.2
XS GIS Cut Line= 3
     1814450.008      464088.281     1814472.143         464100.
     1814582.821      464129.948
#Sta/Elev= 18
       0  924.88     8.4  920.91    16.7  917.03      25  913.96    34.6   911.7
    36.6   911.5    44.2  910.73    51.6  911.55    53.7  911.78    63.3  915.36
    72.8   920.3    82.4  924.82    91.9  928.58   101.5   932.1     111   935.6
   120.6  939.26   130.2  943.16   139.7  947.02
#Mann= 3 , 0 , 0
       0      .1       0    36.6    .045       0    51.6      .1       0
Bank Sta=36.6,51.6
XS Rating Curve= 0 ,0
Exp/Cntr=0.3,0.1

Type RM Length L Ch R = 1 ,6703.1  ,235.8,229.9,223.7
XS GIS Cut Line= 4
     1814361.466      464271.875     1814418.758      464316.146
     1814478.654      464342.187     1814551.571      464353.906
#Sta/Elev= 26
       0  920.95       9  917.34    18.1  913.89    27.2  910.95    36.2  908.58
    45.2  907.16    54.3  907.32    63.4  907.28    72.4  905.95    81.7   904.2
    85.4  903.75    91.1  903.06   100.4  902.68  104.74  903.32   109.7  904.29
     119  908.13   128.4  912.71   137.7  917.14     147  921.45   156.2  925.66
   165.4  929.76   174.6  933.72   183.9  937.56   193.1  941.36   202.3  945.16
   211.6  948.89
#Mann= 3 , 0 , 0
       0      .1       0    91.1    .045       0  104.74      .1       0
Bank Sta=91.1,104.74
XS Rating Curve= 0 ,0
Exp/Cntr=0.3,0.1

Type RM Length L Ch R = 1 ,6473.2  ,182.8,186.4,190.1
XS GIS Cut Line= 3
     1814308.081      464520.573      1814357.56      464540.104
      1814476.05      464558.333
#Sta/Elev= 22
       0  905.61     8.9  903.02    17.7  900.28    26.6  897.99    35.5   896.4
    44.3  895.22    53.2  893.92    62.4   892.5      67   892.1    71.6  891.71
    80.9  891.95      82  892.41    90.1  895.81    99.3   903.7   108.5  911.95
   117.8  918.86     127  924.99   136.2  930.97   145.4   936.9   154.6  942.78
   163.9  948.56   173.1  954.31
#Mann= 3 , 0 , 0
       0      .1       0      67    .045       0      82      .1       0
Bank Sta=67,82
XS Rating Curve= 0 ,0
Exp/Cntr=0.3,0.1

Type RM Length L Ch R = 1 ,6286.7  ,263.6,264.5,264.7
XS GIS Cut Line= 3
     1814291.154      464641.666     1814322.404      464717.187
     1814423.966      464751.041
#Sta/Elev= 23
       0  896.61     9.1  895.64    18.2  894.63    27.2  893.61    36.3  892.76
    45.4  891.86    54.5  890.86    63.6     890    72.6  889.02    81.7  887.78
    91.5  886.34      96  885.83   101.2  885.25   110.9   886.1     111  886.16
   120.7  891.56   130.4  901.96   140.1  912.31   149.9  920.72   159.6  928.52
   169.3  935.94     179  942.19   188.8  946.86
#Mann= 3 , 0 , 0
       0      .1       0      96    .045       0     111      .1       0
Bank Sta=96,111
XS Rating Curve= 0 ,0
Exp/Cntr=0.3,0.1

Type RM Length L Ch R = 1 ,6022.2  ,232.3,231.9,231.4
XS GIS Cut Line= 2
     1814117.977      464908.593     1814314.591      464978.906
#Sta/Elev= 25
       0  912.76     9.5  906.52      19  900.32    28.5  894.25      38  888.52
    47.5  883.97      57  881.49    66.4  880.54    71.4  880.22    75.9  879.94
    85.4  880.08    86.4  880.23    94.9  881.49   104.4   882.2   113.9  882.21
   123.4  882.11   132.9  882.16   142.4  882.41   151.9  882.88   161.4   883.5
   170.8  884.05   180.3  884.69   189.8  885.52   199.3  886.44   208.8   887.6
#Mann= 3 , 0 , 0
       0      .1       0    71.4    .045       0    85.4      .1       0
Bank Sta=71.4,85.4
XS Rating Curve= 0 ,0
Exp/Cntr=0.3,0.1

Type RM Length L Ch R = 1 ,5790.3  ,189,198.2,204.7
XS GIS Cut Line= 3
     1814043.758      465128.646     1814145.321        465162.5
     1814233.862      465149.479
#Sta/Elev= 25
       0  902.26     9.7  897.96    19.5  892.79    29.2   887.2    38.9  880.78
    48.7  875.34    54.5  873.92    58.4  872.97    68.1  872.68    69.5  872.78
   73.52  873.04    77.9  873.39    87.6  874.34    97.3  875.19   107.1  875.91
     116  876.59     125  877.17   133.9  877.56   142.8  877.84   151.8   878.2
   160.8  878.74   169.7  879.34   178.6  880.01   187.6  880.83   196.6  881.71
#Mann= 3 , 0 , 0
       0      .1       0    58.4    .045       0   73.52      .1       0
Bank Sta=58.4,73.52
XS Rating Curve= 0 ,0
Exp/Cntr=0.3,0.1

Type RM Length L Ch R = 1 ,5592.1  ,94.7,57.3,20.1
XS GIS Cut Line= 3
     1813994.279      465300.521     1814014.244      465316.146
      1814109.73      465387.326
#Sta/Elev= 19
       0   878.3     8.4  877.08    16.9  875.18    25.4  872.84    34.5  870.28
    39.3  869.71    43.7  869.18    52.8  868.84    54.3  868.87      62  869.02
    71.2  869.47    80.3  869.83    89.5  870.02    98.6  870.65   107.8  874.97
     117  885.07   126.1   895.4   135.3  903.88   144.4  911.01
#Mann= 3 , 0 , 0
       0      .1       0    39.3    .045       0    54.3      .1       0
Bank Sta=39.3,54.3
XS Rating Curve= 0 ,0
Exp/Cntr=0.3,0.1

Type RM Length L Ch R = 1 ,5534.9  ,34.6,27,30.3
XS GIS Cut Line= 4
     1813958.689      465391.666     1813987.334      465411.632
     1814039.418      465357.812     1814087.161      465396.875
#Sta/Elev= 22
       0  873.57    4.35  872.06    8.75  870.75    13.1  869.65   17.45  868.75
   22.15  868.36    26.8  868.18    31.5  868.11    33.2   868.1    36.2  868.08
    40.7  868.22   40.85  868.22   45.55  868.33    50.2  868.48    54.9  868.89
    59.3  869.23    63.7  869.38    68.1  869.63   72.55  873.56   76.95  881.46
   81.35  891.72   85.75  900.52
#Mann= 3 , 0 , 0
       0      .1       0    33.2    .045       0    40.7      .1       0
Bank Sta=33.2,40.7
XS Rating Curve= 0 ,0
Skew Angle= 60
Exp/Cntr=0.3,0.1

Type RM Length L Ch R = 1 ,5507.9  ,47.4,93.7,129.8
XS GIS Cut Line= 4
     1813934.383      465402.951     1813989.939      465440.277
     1814042.022      465386.458     1814089.765      465425.521
#Sta/Elev= 25
       0  874.93     4.8  873.23    9.55  871.63   14.35   870.3    19.1  869.25
    23.9  868.38    28.7  867.49   33.45  866.84   38.15  867.37    42.8  867.64
    47.5  867.78   51.25  867.84    52.2  867.85   56.85  868.05   58.75  868.14
   61.55  868.28   66.25  868.54    70.9  868.75    75.3  870.04    79.7  875.43
   84.15  884.36   88.55  893.98   92.95  902.39   97.35  910.13  101.75  917.38
#Mann= 3 , 0 , 0
       0      .1       0   51.25    .045       0   58.75      .1       0
Bank Sta=51.25,58.75
XS Rating Curve= 0 ,0
Skew Angle= 60
Exp/Cntr=0.3,0.1

Type RM Length L Ch R = 1 ,5414.2  ,160,159.2,158.3
XS GIS Cut Line= 2
     1813891.848      465422.916     1814036.814       465541.84
#Sta/Elev= 23
       0  876.91     9.4  875.36    18.8  873.99    28.1  872.76    37.5  871.44
    46.9  870.19    56.2  868.86    65.6  867.46      75  866.08    84.4  865.19
    87.8  865.12    93.8     865   102.8  866.99   103.1  867.06   112.5  874.11
   121.9  883.25   131.2   891.5   140.6  898.46     150  905.42   159.4  912.57
   168.8  919.88   178.1  927.21   187.5  934.53
#Mann= 3 , 0 , 0
       0      .1       0    84.4    .045       0   102.8      .1       0
Bank Sta=84.4,102.8
XS Rating Curve= 0 ,0
Exp/Cntr=0.3,0.1

Type RM Length L Ch R = 1 ,5255    ,135.7,133.7,131.4
XS GIS Cut Line= 2
     1813814.591      465566.146     1813950.008      465667.708
#Sta/Elev= 22
       0  870.67     9.4  869.11    18.8  867.58    28.2  866.12    37.6   864.8
      47  863.53    56.4  862.65    65.8  862.34    75.2  862.21    84.6  861.71
    89.4  861.64      94  861.57   99.49  862.83   103.4  863.92   104.4  864.61
   112.8  870.36   122.2  879.74   131.7  888.37   141.1  896.59   150.5  904.49
   159.9  911.78   169.3  918.08
#Mann= 3 , 0 , 0
       0      .1       0    84.6    .045       0   99.49      .1       0
Bank Sta=84.6,99.49
XS Rating Curve= 0 ,0
Exp/Cntr=0.3,0.1

Type RM Length L Ch R = 1 ,5121.3  ,89.5,90.1,91
XS GIS Cut Line= 4
     1813773.619      465675.392     1813796.189      465721.399
     1813848.272      465753.517     1813926.397      465751.781
#Sta/Elev= 24
       0  864.92     8.5  863.65    17.1  862.65    25.6  861.81    34.2  861.02
    42.7  860.21    51.2  859.39      60  858.64    68.7  857.84    77.5     857
    83.7  856.49    86.2  856.28      95  856.36    98.7  857.12   103.7  858.15
   112.4   861.5   122.2  866.52     132  871.81   141.7  877.02   151.5  882.19
   161.3  887.38     171   892.5   180.8  897.45   190.6  902.17
#Mann= 3 , 0 , 0
       0      .1       0    83.7    .045       0    98.7      .1       0
Bank Sta=83.7,98.7
XS Rating Curve= 0 ,0
Exp/Cntr=0.3,0.1

Type RM Length L Ch R = 1 ,5031.2  ,35.4,34.6,33.7
XS GIS Cut Line= 2
     1813727.786      465782.291     1813889.244       465889.93
#Sta/Elev= 23
       0  857.48     9.7  856.74    19.4  856.24    29.1  856.03    38.8  855.86
    48.5  855.23    57.8  854.13    58.2  854.08    67.9   853.6    72.8  853.75
    77.6   853.9    87.3  854.88      97  855.75   106.7  855.99   116.4  856.35
   126.1  856.63   135.8  856.95   145.5   857.3   155.2  857.67   164.9  858.06
   174.6  858.55   184.4  859.02     194  859.52
#Mann= 3 , 0 , 0
       0     .07       0    58.2    .045       0    77.6      .1       0
Bank Sta=58.2,77.6
XS Rating Curve= 0 ,0
Exp/Cntr=0.3,0.1

Type RM Length L Ch R = 1 ,4996.6  ,32.6,32.5,32.4
XS GIS Cut Line= 3
     1813676.397      465794.315     1813808.515      465875.173
     1813873.619      465913.368
#Sta/Elev= 27
       0  857.79     9.7  856.83    19.4  855.98      29  855.43    38.7  855.08
    48.4   854.8    58.1  854.53    67.8  854.49    77.4  854.53    87.1  854.03
    94.7  853.13    96.8  852.88   106.5  852.78   109.7  853.26   116.2  854.22
   125.8  855.54   135.5  855.92   145.2  855.88   154.9  855.91   164.3  856.09
   173.8  856.38   183.2  856.68   192.6  857.05   202.1   857.4   211.5  857.77
   220.9  858.18   230.4  858.59
#Mann= 3 , 0 , 0
       0     .07       0    94.7    .045       0   109.7     .07       0
Bank Sta=94.7,109.7
XS Rating Curve= 0 ,0
Exp/Cntr=0.3,0.1

Type RM Length L Ch R = 1 ,4964.1  ,73.8,75.9,77.9
XS GIS Cut Line= 3
     1813651.223      465816.885      1813788.55      465900.347
     1813853.654      465938.541
#Sta/Elev= 28
       0  856.77     9.4  855.58    18.9  854.56    28.4   854.2    37.8  854.07
    47.3   853.9    56.7  853.68    66.2   853.5    75.6  853.51    85.1  852.97
    94.5  851.96   100.5  851.56     104  851.32   113.4  851.48   115.5  851.74
   122.9  852.66   132.3  854.22   141.8  854.75   151.2  854.94   160.7  854.86
   170.1  854.96   179.6  855.33     189  855.66   198.4  855.94   207.9  856.15
   217.3  856.41   226.8  856.78   236.2  857.24
#Mann= 3 , 0 , 0
       0     .07       0   100.5    .045       0   115.5     .07       0
Bank Sta=100.5,115.5
XS Rating Curve= 0 ,0
Exp/Cntr=0.3,0.1

Type RM Length L Ch R = 1 ,4888.2  ,94.3,98.7,104.7
XS GIS Cut Line= 2
     1813621.015      465876.909     1813818.064      466021.875
#Sta/Elev= 28
       0  854.68     9.8  854.08    19.6  853.49    29.4  853.06    39.1  852.83
    48.9  852.67    58.7  852.51    68.5  852.07    78.3  851.01      87  849.94
    88.1  849.81    97.8  849.27     102  849.68   107.6  850.22   117.4  852.02
   127.2   853.4     137  853.88   146.8  854.14   156.6  853.98   166.4  854.22
   176.1  854.54   185.9   855.1   195.7  855.45   205.5  855.34   215.3  855.32
   225.1  855.76   234.8  856.17   244.6  856.69
#Mann= 3 , 0 , 0
       0     .07       0      87    .045       0     102      .1       0
Bank Sta=87,102
XS Rating Curve= 0 ,0
Exp/Cntr=0.3,0.1

Type RM Length L Ch R = 1 ,4789.5  ,136.8,139.7,139.9
XS GIS Cut Line= 4
     1813581.084      465959.375     1813606.258      465978.472
     1813631.432      466005.382     1813668.758      466066.146
#Sta/Elev= 19
       0  853.66     7.9  853.35    15.8  853.07    23.7   852.7    31.6  851.59
    40.8  849.57    47.2  848.35      50  847.82    59.2  849.02    62.2  850.61
    68.4  853.89    77.4  862.62    86.3  870.18    95.2  876.42   104.1  882.27
     113  888.18   121.9     894   130.8  899.72   139.8  905.28
#Mann= 3 , 0 , 0
       0      .1       0    47.2    .045       0    59.2      .1       0
Bank Sta=47.2,59.2
XS Rating Curve= 0 ,0
Exp/Cntr=0.3,0.1

Type RM Length L Ch R = 1 ,4649.8  ,168.3,166.6,165.7
XS GIS Cut Line= 4
     1813486.466      466044.444     1813497.751      466061.805
     1813519.453      466091.319     1813568.064      466134.722
#Sta/Elev= 16
       0  854.09     6.9  853.31    13.8  851.56    20.7  848.95    29.9   845.5
      39  844.31    44.9  845.63    48.2  846.37    57.3  852.32    66.6  860.35
      76  867.95    85.3  875.01    94.6  881.82   103.9  888.42   113.2   894.8
   122.5  901.01
#Mann= 3 , 0 , 0
       0      .1       0    29.9    .045       0    44.9      .1       0
Bank Sta=29.9,44.9
XS Rating Curve= 0 ,0
Exp/Cntr=0.3,0.1

Type RM Length L Ch R = 1 ,4483.1  ,171.2,172.4,173.5
XS GIS Cut Line= 2
     1813344.105      466136.458     1813410.078      466215.451
#Sta/Elev= 14
       0  848.86     9.4  847.48    18.7  843.49    27.6  839.59    28.1  839.37
    37.4  838.35    42.6  839.39    46.8  840.23    56.1  847.52    65.5  856.91
    74.8  865.18    84.2  872.58    93.6  880.11   102.9  887.42
#Mann= 3 , 0 , 0
       0      .1       0    28.1    .045       0    42.6      .1       0
Bank Sta=28.1,42.6
XS Rating Curve= 0 ,0
Exp/Cntr=0.3,0.1

Type RM Length L Ch R = 1 ,4310.8  ,169.8,169.6,168.9
XS GIS Cut Line= 2
     1813200.008      466226.736       1813257.3      466303.125
#Sta/Elev= 15
       0  844.12     9.6  842.86    19.1  839.25   25.95  836.81    28.6  835.79
    28.8  835.79    38.2  836.02   41.81  837.88    43.8  838.84    47.7  840.81
    57.3  849.08    66.8  857.92    76.4  865.93    85.9  873.73    95.5  881.35
#Mann= 3 , 0 , 0
       0      .1       0   25.95    .045       0   41.81      .1       0
Bank Sta=25.95,41.81
XS Rating Curve= 0 ,0
Exp/Cntr=0.3,0.1

Type RM Length L Ch R = 1 ,4141.2  ,223,221.8,219.9
XS GIS Cut Line= 2
       1813069.8      466336.111     1813122.751      466403.819
#Sta/Elev= 12
       0  841.74     9.6  840.28    19.1  836.64    25.6  833.78    28.6  832.46
    38.2  832.36    40.6   833.6    47.8  837.31    57.3  846.78    66.8  857.87
    76.4  867.74      86  876.29
#Mann= 3 , 0 , 0
       0      .1       0    25.6    .045       0    40.6      .1       0
Bank Sta=25.6,40.6
XS Rating Curve= 0 ,0
Exp/Cntr=0.3,0.1

Type RM Length L Ch R = 1 ,3919.4  ,163.8,163.8,163.2
XS GIS Cut Line= 2
     1812896.189      466476.736     1812952.612      466539.236
#Sta/Elev= 12
       0  837.87     9.4  836.65    18.7  832.71    28.1  827.66    28.7  827.47
    37.4  824.71    43.7  826.12    46.8  826.82    56.1  834.78    65.5  845.05
    74.8  852.97    84.2  859.68
#Mann= 3 , 0 , 0
       0      .1       0    28.7    .045       0    43.7      .1       0
Bank Sta=28.7,43.7
XS Rating Curve= 0 ,0
Exp/Cntr=0.3,0.1

Type RM Length L Ch R = 1 ,3755.6  ,195.8,193.5,191.3
XS GIS Cut Line= 2
     1812784.209      466591.319     1812848.446      466660.764
#Sta/Elev= 13
       0  832.25     9.5  830.42    18.9  824.57    28.4  818.38    35.5  816.46
    37.8  815.84    47.3  816.76    50.5  818.62    56.8  822.29    66.2  833.72
    75.7  843.56    85.1  851.25    94.6  858.27
#Mann= 3 , 0 , 0
       0      .1       0    35.5    .045       0    47.3      .1       0
Bank Sta=35.5,47.3
XS Rating Curve= 0 ,0
Exp/Cntr=0.3,0.1

Type RM Length L Ch R = 1 ,3562.1  ,127.9,127.5,133
XS GIS Cut Line= 2
     1812640.112      466727.604     1812731.258      466808.333
#Sta/Elev= 16
       0  818.89     9.4  818.28    18.7   817.5    28.1  816.02    37.5   813.4
    46.8  810.58    48.7   810.3    56.2  809.21    63.7  809.79    65.6  809.94
    74.9  815.86    84.3  826.67    93.7  837.19     103  845.35   112.4  852.86
   121.8  860.18
#Mann= 3 , 0 , 0
       0      .1       0    48.7    .045       0    65.6      .1       0
Bank Sta=48.7,65.6
XS Rating Curve= 0 ,0
Exp/Cntr=0.3,0.1

Type RM Length L Ch R = 1 ,3434.6  ,18,51.7,104.3
XS GIS Cut Line= 3
     1812493.237       466747.44     1812578.307      466823.829
     1812600.876      466884.593
#Sta/Elev= 22
       0  829.31     9.5  822.34    19.1  815.36    28.6  810.63    38.1  809.18
    47.6  809.52    57.2  809.71    66.7   809.5    76.2  808.07    85.8   805.9
    94.9  804.54    95.3  804.48   104.8  805.33   109.9  807.49   114.3  809.36
   123.6  817.68   132.8  826.95   142.1  834.52   151.4  841.52   160.6  847.08
   169.9  851.26   179.2  854.98
#Mann= 3 , 0 , 0
       0      .1       0    85.8    .045       0   104.8      .1       0
Bank Sta=85.8,104.8
XS Rating Curve= 0 ,0
Exp/Cntr=0.3,0.1

Type RM Length L Ch R = 1 ,3383    ,64,75.3,64.4
XS GIS Cut Line= 4
     1812462.161       466760.59     1812548.098      466817.014
     1812486.466      466883.854     1812544.626      466926.389
#Sta/Elev= 26
       0  832.75     4.7  826.45    9.35  820.46      14     814    18.7  808.97
   23.35  807.46   28.05  807.46    32.7  807.86    37.4  808.07   42.05  807.65
   46.75  806.22    51.4   804.5   55.95  804.05    60.5  803.44   65.05  803.21
   74.15   802.3   87.75  801.93    92.3  802.36   96.85  802.25  101.35  805.78
  105.85  811.43   114.9  824.78   119.4  831.86   123.9  838.68   128.4  844.93
   132.9  849.98
#Mann= 3 , 0 , 0
       0      .1       0   65.05    .045       0   74.15      .1       0
Bank Sta=65.05,74.15
XS Rating Curve= 0 ,0
Skew Angle= 60
Exp/Cntr=0.3,0.1

Type RM Length L Ch R = 1 ,3307.7  ,146.3,96.5,43.3
XS GIS Cut Line= 4
     1812398.793      466773.611      1812484.73      466830.034
     1812423.098      466896.875     1812481.258      466939.409
#Sta/Elev= 28
       0  855.58     4.7  849.66    9.35  843.68      14  837.93    18.7  831.94
   23.35  825.38   28.05   816.5    32.7  807.94    37.4  803.48   42.05  802.44
   46.75   803.3    51.4  803.76    60.5  801.44   65.05  799.89    69.6  798.02
   70.05  797.91   74.15  796.86    78.7  796.32   87.75  796.39    92.3  796.11
   96.85  795.68  101.35   797.6  105.85  798.93   114.9  800.07   119.4  801.39
   123.9  803.88   128.4  808.54   132.9  813.58
#Mann= 3 , 0 , 0
       0      .1       0   70.05    .045       0    78.7      .1       0
Bank Sta=70.05,78.7
XS Rating Curve= 0 ,0
Skew Angle= 60
Exp/Cntr=0.3,0.1

Type RM Length L Ch R = 1 ,3211.2  ,102,104.5,106.4
XS GIS Cut Line= 4
     1812340.633      466899.479     1812363.203      466913.368
     1812412.682      466942.014     1812512.508      466974.132
#Sta/Elev= 23
       0  817.54     8.8  810.72    17.7  803.71    26.5  798.29      36  794.55
    45.6  792.87    48.2  792.68    55.1  792.19    63.2  792.96    64.6  793.09
    74.1  794.98    83.7  796.38    93.2   797.4   102.7  798.47   112.3  799.61
   121.8  801.05   131.3  803.95   140.9  808.71   150.4  814.58   159.9  821.39
   169.5  828.59     179  835.13   188.5  841.02
#Mann= 3 , 0 , 0
       0      .1       0    45.6    .045       0    63.2      .1       0
Bank Sta=45.6,63.2
XS Rating Curve= 0 ,0
Exp/Cntr=0.3,0.1

Type RM Length L Ch R = 1 ,3106.7  ,118.3,119.5,120.8
XS GIS Cut Line= 2
     1812289.418      466984.548     1812454.348      467102.604
#Sta/Elev= 24
       0  812.83     9.7  807.59    19.3  803.04      29  799.42    38.6  796.24
    48.3  792.38    51.1  791.73      58  790.14    66.1  789.99    67.6  789.96
    77.3  790.59    86.9  791.22    96.6  791.93   106.2  792.74   115.9  793.28
   125.6  793.64   135.2  793.84   144.9  793.99   154.5  794.68   164.2  797.36
   173.8  802.63   183.5  809.51   193.2   816.6   202.8  823.82
#Mann= 3 , 0 , 0
       0      .1       0    51.1    .045       0    67.6     .08       0
Bank Sta=51.1,67.6
XS Rating Curve= 0 ,0
Exp/Cntr=0.3,0.1

Type RM Length L Ch R = 1 ,2987.2  ,133.4,135.1,136.1
XS GIS Cut Line= 2
     1812247.751      467096.527     1812392.716      467212.847
#Sta/Elev= 23
       0  806.99     9.8   800.6    19.6  794.52    29.4  789.69    34.8  788.38
    39.1  787.34    48.9  787.03    49.8  787.08   53.68  787.27    58.7  787.59
    68.5  788.12    78.3  788.52      88  788.86    97.8  789.27   107.6  789.69
   117.4  790.13   127.2  790.89     137  794.02   146.7  799.44   156.5  806.15
   166.3  813.31   176.1  819.96   185.9  826.82
#Mann= 3 , 0 , 0
       0      .1       0    39.1    .045       0   53.68     .08       0
Bank Sta=39.1,53.68
XS Rating Curve= 0 ,0
Exp/Cntr=0.3,0.1

Type RM Length L Ch R = 1 ,2852.1  ,125.4,122.1,119
XS GIS Cut Line= 4
     1812151.397      467182.465      1812172.23      467205.902
     1812254.696      467278.819     1812305.911      467303.993
#Sta/Elev= 25
       0  817.72     7.8  811.67    15.7  805.12    23.5  796.93    31.4  789.38
    40.5  784.46    41.9  784.29    49.7  783.36    56.9  783.76    58.9  783.87
      68  784.39    77.2  784.66    86.4  784.93    95.6   785.2   104.7  785.47
   113.9  785.74   123.1  786.06   132.3  786.49   141.4  788.19     151  792.07
   160.5  797.28     170  802.46   179.5  807.58     189  812.74   198.5  817.95
#Mann= 3 , 0 , 0
       0      .1       0    41.9    .045       0    56.9     .08       0
Bank Sta=41.9,56.9
XS Rating Curve= 0 ,0
Exp/Cntr=0.3,0.1

Type RM Length L Ch R = 1 ,2730.1  ,110.1,111,110.6
XS GIS Cut Line= 4
      1812074.14      467289.236     1812096.709      467303.993
     1812177.439       467358.68     1812219.973      467435.069
#Sta/Elev= 25
       0  809.43       9  800.05      18  790.93      27  783.83    34.2  781.21
    36.7   780.3    46.5  780.14    49.2  780.32    56.2  780.77      66  781.07
    75.7  781.52    85.5  782.09    95.2  782.61     105   783.1   114.7  783.51
   124.5  783.99   134.2  785.28   143.9  788.28   153.6  792.44   163.3   797.3
     173   802.1   182.8   806.9   192.5  811.05   202.2   815.3   211.9  819.24
#Mann= 3 , 0 , 0
       0      .1       0    34.2    .045       0    49.2     .08       0
Bank Sta=34.2,49.2
XS Rating Curve= 0 ,0
Exp/Cntr=0.3,0.1

Type RM Length L Ch R = 1 ,2619.1  ,161.4,170.3,174.5
XS GIS Cut Line= 4
     1812014.244      467376.041      1812038.55      467398.611
     1812088.897      467431.597      1812167.89      467488.021
#Sta/Elev= 24
       0  802.41     8.3  796.68    16.6  791.06    24.9  785.04    33.2  779.91
    41.8  777.01    42.3     777    50.4  776.77    57.3  777.18      59  777.28
    67.6  777.94    76.2  778.93    84.8  780.63    93.4  782.66   103.1     785
   112.8  787.44   122.5  790.24   132.2  793.56   141.9  798.22   151.6  804.08
   161.3   810.3     171  816.54   180.7  822.61   190.4  828.54
#Mann= 3 , 0 , 0
       0      .1       0    42.3    .045       0      59     .06       0
Bank Sta=42.3,59
XS Rating Curve= 0 ,0
Exp/Cntr=0.3,0.1

Type RM Length L Ch R = 1 ,2448.8  ,154.4,158.1,167
XS GIS Cut Line= 4
     1811939.591      467515.798     1811946.536      467538.368
     1811985.425      467575.565     1812074.834      467616.364
#Sta/Elev= 22
       0  786.81     7.9  784.91    15.7  782.36    23.6  778.63    28.5  776.34
    32.6  774.43    41.6  772.92    43.5  772.95    50.5  773.06    59.5  773.77
    68.5  774.65    77.4  775.31    87.3  775.86    97.1  776.34   106.9  776.86
   116.7  777.46   126.6  778.31   136.4  780.71   146.2  785.87     156  792.82
   165.9  800.16   175.7  807.45
#Mann= 3 , 0 , 0
       0      .1       0    32.6    .045       0    50.5     .08       0
Bank Sta=32.6,50.5
XS Rating Curve= 0 ,0
Exp/Cntr=0.3,0.1

Type RM Length L Ch R = 1 ,2290.7  ,145,127.2,109.3
XS GIS Cut Line= 2
     1811811.987      467564.409     1811900.529      467755.382
#Sta/Elev= 25
       0  781.67     9.6  776.65    19.1  773.44    28.7  771.55    38.3  770.36
    47.8  769.92    57.4  769.66      67  769.56    76.6  769.36    86.1  768.96
    95.7  768.13   105.2  767.16   113.5  766.86   114.8  766.81   124.4  767.31
   128.5  768.13     134  769.24   143.5  770.75   153.1  771.73   162.7  773.89
   172.2  778.03   181.8  783.68   191.4  790.36   200.9  797.55   210.5  803.32
#Mann= 3 , 0 , 0
       0     .08       0   105.2    .045       0   124.4     .06       0
Bank Sta=105.2,124.4
XS Rating Curve= 0 ,0
Exp/Cntr=0.3,0.1

Type RM Length L Ch R = 1 ,2163.5  ,197,204.3,210.1
XS GIS Cut Line= 4
     1811704.348      467732.812     1811745.147      467744.965
     1811811.119      467770.139     1811897.057      467821.354
#Sta/Elev= 27
       0  792.13     8.5  785.33      17  779.01    25.5   774.1    34.1  770.97
    42.6  768.47    51.4  766.59    60.2  765.63      69  765.56    72.4  765.74
    77.9  766.02    86.7  766.08    87.4  766.12    95.5  766.62   104.4  767.71
   113.2  768.83   122.3  769.71   131.4  769.98   140.5  770.85   149.6  774.66
   158.7  781.28   167.8  788.39   176.8  794.18   185.9  799.79     195  805.77
   204.1     812   213.2  817.72
#Mann= 3 , 0 , 0
       0     .06       0    72.4    .045       0    87.4     .06       0
Bank Sta=72.4,87.4
XS Rating Curve= 0 ,0
Exp/Cntr=0.3,0.1

Type RM Length L Ch R = 1 ,1959.2  ,191.2,188.3,185.5
XS GIS Cut Line= 4
     1811617.543      467852.604     1811634.036      467879.514
     1811733.862      467954.166     1811812.855      467997.569
#Sta/Elev= 30
       0  788.91     7.9  783.46    15.8  777.57    23.7  771.44    31.6  766.12
    41.2  761.81    50.7  760.68    60.3  760.77    69.9  761.08    79.5  761.56
    89.1  761.99    98.7  762.23   108.3  762.13   117.9  761.66     126  761.01
   127.4   760.9     137  760.34     141  761.05   146.6  762.04   156.2  767.26
   165.2  775.04   174.2  783.42   183.2  790.82   192.3  797.57   201.3   804.5
   210.3  811.22   219.3  817.07   228.3  822.42   237.3   827.9   246.4  833.91
#Mann= 3 , 0 , 0
       0     .06       0     126    .045       0     141      .1       0
Bank Sta=126,141
XS Rating Curve= 0 ,0
Exp/Cntr=0.3,0.1

Type RM Length L Ch R = 1 ,1770.9  ,171.4,176,181.2
XS GIS Cut Line= 4
     1811518.584      468042.708      1811542.89      468058.333
      1811663.55      468126.041     1811722.578      468134.722
#Sta/Elev= 28
       0   781.4     9.6  775.25    19.3  767.41    28.9   759.8    38.1  755.94
    47.3  755.24    56.6  755.34    65.8  755.69      75  756.06    84.2  756.27
    93.5  756.35   102.7  756.35   111.9  756.18   121.1  755.78   129.2  755.15
   130.4  755.06   139.6  754.58   144.2  754.84   148.8   755.1     158  759.33
   167.2  768.26   175.8  779.35   184.3  791.03   192.8  801.95   201.4  810.33
   209.9  816.83   218.4  822.44   226.9  827.73
#Mann= 3 , 0 , 0
       0     .08       0   129.2    .045       0   148.8      .1       0
Bank Sta=129.2,148.8
XS Rating Curve= 0 ,0
Exp/Cntr=0.3,0.1

Type RM Length L Ch R = 1 ,1594.9  ,150,148.4,145.2
XS GIS Cut Line= 4
     1811445.668      468154.904     1811457.821      468185.286
     1811562.855      468272.092     1811594.973      468320.703
#Sta/Elev= 27
       0  773.37     8.2  768.94    16.4  763.89    24.5  758.96    32.7  755.54
    42.5  753.29    52.2  752.16    61.9   751.4    71.6  750.98    81.4     751
    91.1  751.53   100.8  752.21   110.6  752.78   120.3  752.98     130  752.76
   139.8  751.76   142.9  751.51   149.5  750.97   157.9  751.58   159.2  751.68
     169  757.17   178.7  768.59   188.4  781.86   198.1  793.61   207.8  802.17
   217.5  808.41   227.2  813.78
#Mann= 3 , 0 , 0
       0     .08       0   142.9    .045       0   159.2      .1       0
Bank Sta=142.9,159.2
XS Rating Curve= 0 ,0
Exp/Cntr=0.3,0.1

Type RM Length L Ch R = 1 ,1446.5  ,154.5,175.7,197.5
XS GIS Cut Line= 2
     1811318.064      468275.564     1811516.848      468418.793
#Sta/Elev= 28
       0  754.11     9.8  751.77    19.6  751.27    29.4   750.4    39.2  749.22
      49  748.26    58.8  747.62    68.6  747.18    78.4   746.8    88.2  746.38
      98  746.14   107.8  746.21   117.6  746.56   127.4  747.24   137.2  747.96
     147  748.27   155.2   747.9   156.8  747.83   166.6  747.02   170.2  748.58
   176.4  751.27   186.2  761.26     196  772.96   205.8  783.61   215.6  792.02
   225.4  797.78   235.2  802.77     245  807.73
#Mann= 3 , 0 , 0
       0     .08       0   156.8    .045       0   170.2      .1       0
Bank Sta=156.8,170.2
XS Rating Curve= 0 ,0
Exp/Cntr=0.3,0.1

Type RM Length L Ch R = 1 ,1270.9  ,173.7,150.9,126.3
XS GIS Cut Line= 4
     1811194.843      468394.142     1811352.786      468488.238
     1811329.348      468518.619     1811391.848      468567.231
#Sta/Elev= 30
       0  763.21     9.7  758.38    19.4  753.89      29   749.9    38.7  746.35
    48.4  743.69    58.1  742.34    67.7  741.95    77.4  741.87   116.1  741.93
   125.8  742.37   135.5  743.24   145.1  743.86   154.8  743.89   164.5  743.71
   174.2  743.31   183.8  742.17   197.4   741.2     203  740.73   212.4  740.53
   222.2  740.71     231  741.34   239.8  743.35   248.6   747.5   257.4   752.7
   266.2  759.67     275  767.26   283.8  774.64   292.6  781.63   301.4  787.65
#Mann= 3 , 0 , 0
       0     .06       0   197.4    .045       0   212.4      .1       0
Bank Sta=197.4,212.4
XS Rating Curve= 0 ,0
Exp/Cntr=0.3,0.1

Type RM Length L Ch R = 1 ,1120    ,153.2,156.3,157.7
XS GIS Cut Line= 2
      1811144.93      468482.032     1811357.126      468604.557
#Sta/Elev= 27
       0  767.68     9.8  763.85    19.6  759.75    29.4  754.44    39.2   746.7
      49  740.15    53.6  739.38    58.8  738.51    68.6  738.64    78.4  739.14
    88.2  739.46      98  739.66   107.8  739.85   117.6  739.98   127.4  739.91
   137.2   739.8     147  739.88   156.8  740.31   166.6  741.13   176.4  741.93
   186.2  742.27     196  742.37   205.8   742.8   215.6  745.34   225.4  751.52
   235.2  761.05     245     771
#Mann= 3 , 0 , 0
       0     .06       0    53.6    .045       0    68.6     .08       0
Bank Sta=53.6,68.6
XS Rating Curve= 0 ,0
Exp/Cntr=0.3,0.1

Type RM Length L Ch R = 1 ,963.7   ,190,188,187.4
XS GIS Cut Line= 4
      1811101.05      468623.654     1811120.147      468643.619
     1811217.369      468709.592     1811335.425      468780.772
#Sta/Elev= 24
       0   758.7     9.2  754.48    18.4  749.03    27.6   742.1    37.4  735.45
    47.2  734.12    51.7  734.39    66.8  735.37    76.6  735.64    86.4  735.73
    96.2   735.7   115.8  735.51   125.5   735.7   135.3  736.17   145.1  736.84
   172.7  738.52   181.9  739.26   191.1  741.52   200.3  746.89     237   772.1
   246.2  777.69   255.4   781.9   264.6  785.42     283  792.24
#Mann= 3 , 0 , 0
       0      .1       0    37.4    .045       0    51.7      .1       0
Bank Sta=37.4,51.7
XS Rating Curve= 0 ,0
Exp/Cntr=0.3,0.1

Type RM Length L Ch R = 1 ,775.7   ,59.3,59.2,58.9
XS GIS Cut Line= 4
     1810989.939      468766.015      1811011.64      468792.925
     1811133.385      468870.507     1811259.253      468866.167
#Sta/Elev= 30
       0  748.34     8.6  744.28    17.3  740.33    25.9  737.19    34.6   734.2
    44.2  731.28   50.53  730.54    53.8  730.22    63.4  730.28    68.3  730.57
    73.1  730.85    82.7  731.19    92.3   731.3   101.9   731.3   130.8   731.6
   140.4  731.57   150.1  731.43   159.7   731.5   169.3  731.89   178.9  732.53
   188.6  733.34   198.3  733.85   227.4  735.05   237.1  735.86   246.8  738.06
   256.4  741.86   266.1     746   275.8   749.7   295.2  756.73   304.9  760.45
#Mann= 3 , 0 , 0
       0     .06       0   50.53    .045       0    68.3     .08       0
Bank Sta=50.53,68.3
XS Rating Curve= 0 ,0
Exp/Cntr=0.3,0.1

Type RM Length L Ch R = 1 ,716.5   ,51.3,52.4,57.6
XS GIS Cut Line= 2
     1810952.612      468823.958     1811200.876      468951.562
#Sta/Elev= 22
       0  746.05    19.2  740.52    28.9  738.46    38.5  736.64    48.1  735.42
    57.8  734.02    67.4  732.02      77  730.25      81  730.04    86.6  729.75
      96  729.75   105.9  730.05   115.5  730.09   134.8  729.93   163.6  729.95
   173.3  730.39   192.5  731.48   202.1  731.87   221.4  732.45   240.6  732.89
   259.9  733.59   279.1  734.06
#Mann= 3 , 0 , 0
       0     .08       0      81    .045       0      96     .08       0
Bank Sta=81,96
XS Rating Curve= 0 ,0
Exp/Cntr=0.3,0.1

Type RM Length L Ch R = 1 ,664     ,76.4,71.2,62.7
XS GIS Cut Line= 2
     1810923.098      468855.425     1811171.362      468983.029
#Sta/Elev= 22
       0  756.21     9.6  749.16    19.2  741.22    28.9  734.58    38.5  731.08
    48.1  729.82    57.8  729.59      77  729.33    86.6  729.05   105.9  728.17
   115.5  727.64   124.7   727.3   134.8  726.96   144.4  726.87     154  727.31
   163.6  728.04   173.3  728.67   192.5  730.16   202.1  730.64   221.4  731.06
   259.9   731.6   279.1  731.99
#Mann= 3 , 0 , 0
       0     .08       0   124.7    .045       0   144.4     .06       0
Bank Sta=124.7,144.4
XS Rating Curve= 0 ,0
Exp/Cntr=0.3,0.1

Type RM Length L Ch R = 1 ,592.8   ,33.1,41.7,51
XS GIS Cut Line= 4
     1810909.209      468937.022     1810952.612      468942.231
     1811068.932      468992.578     1811187.855      469018.619
#Sta/Elev= 24
       0  756.79     8.7  749.86    17.5  742.74    26.2  735.98      35  730.74
    43.7  728.17    53.5  727.54    92.5  726.92   102.2  726.52   121.7  724.94
   125.7  724.84   131.5   724.7   140.7  725.11     151  726.16   170.5  728.98
   179.8  729.59   198.6  729.81   217.3  731.13   226.6  731.56     236   731.7
   254.7   731.8   264.1  732.01   273.5  732.38   292.2  733.42
#Mann= 3 , 0 , 0
       0     .06       0   125.7    .045       0   140.7     .06       0
Bank Sta=125.7,140.7
XS Rating Curve= 0 ,0
Exp/Cntr=0.3,0.1

Type RM Length L Ch R = 1 ,551.1   ,17.6,16.8,16.9
XS GIS Cut Line= 5
     1810918.107      468949.067     1810941.979      468959.049
     1810997.968       468998.98     1811031.822      469032.834
     1811088.246      469064.952
#Sta/Elev= 25
       0  747.17     8.6  740.16    17.2  733.65    25.9  728.97    35.7  727.41
    45.5  726.95    55.4  726.72    65.2  726.44      75  726.21    84.8  725.56
    94.6  724.37    99.1  723.98   104.2  723.54   113.8  723.67   114.1   723.7
   123.4  724.68     133  726.26   142.5  727.62   151.8  728.32   161.1   728.7
   170.4  729.04   179.6  729.35   188.9  729.74   198.2  730.16   207.4  730.47
#Mann= 3 , 0 , 0
       0      .1       0    99.1    .045       0   114.1     .06       0
Bank Sta=99.1,114.1
XS Rating Curve= 0 ,0
Exp/Cntr=0.3,0.1

Type RM Length L Ch R = 1 ,534.3   ,31.8,30.7,27.6
XS GIS Cut Line= 5
     1810906.822      468961.219     1810930.694      468971.202
     1810986.683      469011.132     1811020.538      469044.987
     1811076.961      469077.105
#Sta/Elev= 25
       0  752.13     8.6  745.08    17.2  737.78    25.9  731.27    35.7   727.6
    45.5  726.42    55.4  725.98    65.2  725.68      75  725.33    84.8  724.73
    94.6   723.7    95.6  723.63   104.2  723.04   110.6  723.13   113.8  723.18
   123.4  724.45     133  726.12   142.5  727.42   151.8  727.83   161.1  728.01
   170.4  728.09   179.6  728.36   188.9  729.05   198.2  729.57   207.4  729.88
#Mann= 3 , 0 , 0
       0      .1       0    95.6    .045       0   113.8     .06       0
Bank Sta=95.6,113.8
XS Rating Curve= 0 ,0
Exp/Cntr=0.3,0.1

Type RM Length L Ch R = 1 ,503.6   ,20.5,28.9,46.1
XS GIS Cut Line= 4
     1810896.362      468989.107     1810923.446      469001.607
     1810990.807      469052.301     1811063.029      469106.468
#Sta/Elev= 26
       0  747.94     7.5  741.66    14.9  735.57    22.4  730.67    29.8  727.05
    39.2  725.06    48.6  724.48    57.9  724.05    67.3   723.4    76.7  722.55
    77.5  722.51      86  722.03    92.5  722.36    95.4  722.51   104.8  723.59
   114.1  725.08   123.2   726.2   132.2  727.14   141.2  727.58   150.2  727.16
   159.3  726.87   168.3   727.2   177.3  728.33   186.4  728.96   195.4  728.77
   204.4  728.69
#Mann= 3 , 0 , 0
       0     .08       0    77.5    .045       0    95.4     .06       0
Bank Sta=77.5,95.4
XS Rating Curve= 0 ,0
Exp/Cntr=0.3,0.1

Type RM Length L Ch R = 1 ,474.7   ,17.9,28.2,18.8
XS GIS Cut Line= 6
      1810892.89      469012.718     1810929.696      469030.774
     1810941.501      469037.024     1810947.751      469075.218
     1810996.362      469105.079      1811049.14      469138.413
#Sta/Elev= 27
       0  740.45     8.2  734.48    16.4  729.29    24.6   725.7    32.8  723.94
      41  723.25    47.7  722.77    54.4  722.27    61.3   721.7      64  721.48
    73.7   721.4    76.3   721.6    83.4  722.14    93.1  723.49   102.6  724.54
   112.1  725.24   121.6  725.95   131.1  726.64   140.6  726.98   150.1   726.7
     159  726.06   167.9  725.92   176.9   726.4   185.8  726.61   194.7  726.94
   203.6  727.27   212.5   727.7
#Mann= 3 , 0 , 0
       0     .06       0    61.3    .045       0    76.3     .06       0
Bank Sta=61.3,76.3
XS Rating Curve= 0 ,0
Exp/Cntr=0.3,0.1

Type RM Length L Ch R = 1 ,446.5   ,37.3,16.8,6.5
XS GIS Cut Line= 6
     1810867.196       469016.19     1810904.001      469034.246
     1810915.807      469040.496     1810922.057       469078.69
     1810970.668      469108.551     1811023.446      469141.885
#Sta/Elev= 27
       0  760.31     8.2  752.12    16.4  744.14    24.6  737.21    32.8  731.04
      41  726.12    47.7  724.04    54.4  722.94      64  721.78    73.2   721.2
    73.7  721.17    83.4  721.09    88.2  721.29    93.1   721.5   102.6  722.76
   112.1  723.91   121.6  724.83   131.1  725.39   140.6  725.92   150.1   725.9
     159  725.83   167.9  725.55   176.9  725.27   185.8  725.45   194.7  725.77
   203.6  726.24   212.5  726.81
#Mann= 3 , 0 , 0
       0     .06       0    73.2    .045       0    88.2     .06       0
Bank Sta=73.2,88.2
XS Rating Curve= 0 ,0
Exp/Cntr=0.3,0.1

Type RM Length L Ch R = 1 ,429.7   ,90,55.9,24.5
XS GIS Cut Line= 4
     1810841.545      469032.313     1810872.795      469054.882
     1810946.579      469100.889      1811111.51      469229.362
#Sta/Elev= 23
       0  775.07     9.6     767    28.9  748.64    38.6  740.02    48.2  732.12
    57.9  725.37    67.5  721.85    77.2  721.01      85  721.19    86.9  721.24
    96.5  722.13   106.2  723.23   115.8  724.18   125.5  724.84     135  725.18
   163.5  724.75     173  725.03     211  726.72   220.5     727     268  727.97
     287  728.27   306.1  728.75   334.6   727.7
#Mann= 3 , 0 , 0
       0     .06       0    67.5    .045       0      85     .06       0
Bank Sta=67.5,85
XS Rating Curve= 0 ,0
Exp/Cntr=0.3,0.1

Type RM Length L Ch R = 1 ,373.8   ,25.1,59.8,52.3
XS GIS Cut Line= 5
     1810672.447      468935.612     1810843.454      469140.473
     1810900.746      469099.674      1811024.01      469179.535
       1811122.1      469281.098
#Sta/Elev= 30
       0  894.88  20.223  878.89  47.164  856.69   60.67  844.31  87.611   818.9
 101.116  806.85 128.057  785.94 141.492  775.05  148.28  768.06 154.998  759.19
 161.715  749.54 168.504  740.63 175.221  732.76 181.939  726.39 188.656  722.32
 207.324  721.82 213.546  721.11 219.627  721.05 225.991  721.27 238.436  721.48
 245.366  722.58 252.296  723.23 300.733  724.98 321.521  726.28 362.251  727.08
 388.909  726.02 395.556   726.1 402.202  727.14 415.496  730.14 442.154  734.52
#Mann= 3 , 0 , 0
       0      .1       0 207.324    .045       0 225.991     .06       0
Bank Sta=207.324,225.991
XS Rating Curve= 0 ,0
Skew Angle= 45
Exp/Cntr=0.3,0.1
